HEC-RAS study Durango.prj: Durango

--- Durango.g18 (geometry) --- (continued)

Type RM Length L Ch R = 4 ,1305.924,,,
BEGIN DESCRIPTION:
E151
END DESCRIPTION:
Bridge Culvert--1,0,-1,-1, 0
Deck Dist Width WeirC Skew NumUp NumDn MinLoCord MaxHiCord MaxSubmerge Is_Ogee
0.01,18.9,1.44,0, 16, 18, , , 0.95, 0, ,,,
   80.35    81.5  81.506  82.562   82.57   82.78  83.108  98.122  98.455  98.905
  98.909  99.939  99.946 100.696 116.985 117.202
 122.659 122.651 123.874 123.923 123.692 123.692 123.693 123.719 123.719  123.72
 123.905 123.898 122.666 122.658 118.155 118.095
   8.375   8.355   8.355   8.338   8.337   8.334 121.626 121.648   8.473   8.477
   8.477   8.487   8.487   8.493   8.639 118.095
  64.111  64.278  81.306  82.456  82.462  83.518  83.526  83.736  84.064  99.078
  99.411  99.861  99.865 100.895 100.902 101.652 117.941 118.158
 117.844  117.89 122.659 122.651 123.874 123.923 123.692 123.692 123.693 123.719
 123.719  123.72 123.905 123.898 122.666 122.658 118.155 118.095
 117.844   8.663   8.375   8.355   8.355   8.338   8.337   8.334 121.626 121.648
   8.473   8.477   8.477   8.487   8.487   8.493   8.639 118.095
BR Coef=-1 , 0 , 0 ,, 0 ,,,0.8,-1,,0,
WSPro=,,,, 1 ,,,, 0 ,,,, 0 ,,,,-1 ,-1 ,-1 , 0 , 0 , 0 , 0 , 0
BC Mult= 1 ,0,81.5,0,83
BC Mult= 3 ,81.5,100,83,101
BC Mult= 1 ,100,300,101,320
BC Design=,, 0 ,, 0 ,,,,,,
BC Use User HTab Curves=0
BC User HTab FreeFlow(D)= 0

Type RM Length L Ch R = 1 ,1295.884,60.31,62.268,64.227
XS GIS Cut Line= 2
529841.7462682324779117.55019448530152.0994712774779141.07591912
#Sta/Elev= 30
       0 138.921   2.031 138.195   5.354     138   6.633 137.471   7.566 135.822
   8.048 134.018   9.051 126.028  11.362 125.825  13.062 125.146  14.065 123.671
  18.514 122.455  46.448 122.132  56.186 122.703  74.237 122.615    83.3  122.21
  83.483 121.785  84.913 118.008  88.915 117.653  98.675 118.039  99.309 120.747
  99.411 122.256 108.244 122.683 144.438 122.874 145.336 122.188 159.961 121.867
 168.837 122.654 207.213 123.003 282.463 124.732 298.337 124.874 311.243 124.275
#Mann= 3 ,-1 , 0
       0      .1       0  83.483    .036       0  99.309      .1       0
#XS Ineff= 2 , 0
            73.7   133.2     107          133.13
Permanent Ineff=
       T       T
#Block Obstruct= 3 ,-1
   57.67   74.32   135.4   106.7  146.48  132.03  170.53  185.64     131
Bank Sta=83.3,99.411
XS Rating Curve= 0 ,0
Exp/Cntr=0.5,0.3

Type RM Length L Ch R = 1 ,1233.615,2.57,2.57,2.57
XS GIS Cut Line= 6
  529840.1537523 4779158.5998097  529890.0445348 4779168.3558333
  529918.8902817 4779188.3848165  529971.4852207 4779197.1830659
    530062.41969 4779224.2449331  530210.4990666        4779266.
#Sta/Elev= 30
       0 127.133   1.783 126.612  11.445 122.136  15.327 121.713   25.57 121.241
  51.711 121.204  68.739 120.788  68.899  117.97  71.424 117.605  75.641 117.444
  80.093 117.713  80.178 118.164    80.9  120.87 161.737 120.707 174.147 121.447
 178.472     121 182.354     121 192.498 121.167 192.945 121.448 208.438 121.641
249.1274121.6271265.0979121.9789288.0556 121.764289.0538122.5084 327.982123.6561
336.9654124.3216354.9323124.6198361.9194124.5699362.9176124.0734 390.866122.3562
#Mann= 4 ,-1 , 0
       0      .1       0   25.57      .1       0  68.899    .036       0
  80.178      .1       0
#XS Ineff= 2 ,-1
   36.34   53.96  124.92   95.15  236.12  130.04
Permanent Ineff=
       T       T
#Block Obstruct= 5 ,-1
  131.72  155.07  129.95  201.76  206.83   131.1     240  248.11  135.24
  290.04  328.46  130.12  362.64  387.67  143.52
Bank Sta=68.739,80.9
XS Rating Curve= 0 ,0
Exp/Cntr=0.5,0.3

Type RM Length L Ch R = 4 ,1232.481,,,
BEGIN DESCRIPTION:
E152
END DESCRIPTION:
Bridge Culvert--1,0,-1,-1, 0
Deck Dist Width WeirC Skew NumUp NumDn MinLoCord MaxHiCord MaxSubmerge Is_Ogee
0.01,2.37,1.44,0, 32, 32, , , 0.95, 0, ,,,
  55.148  55.545  65.124  67.026  68.161  68.259  68.261  68.461   68.47  68.679
  71.722  73.453  73.716  74.453  75.053  75.252  75.793  77.553  78.051  79.555
  79.848  80.866  81.197   81.84  81.845  81.907  81.919  83.901  87.133   87.85
 102.175 102.559
  117.74 117.866 120.905 120.898 120.951 120.955 121.071 121.083 122.069 122.079
  122.22 122.301 122.306 122.322 122.335 122.337 122.318 122.255 122.237 122.175
 122.163 122.085  122.06 122.012 121.006 121.001 120.864 120.494   120.4 120.379
 116.291 116.181
  117.74  40.529  40.436  40.417  40.406   55.42  55.799  86.649   88.14   120.4
 120.591 120.648 120.657  120.66 120.662 120.663 120.665 120.602 120.584  120.53
 120.493 120.363  40.594  40.594  40.594  40.594  40.594  40.594  40.594  40.594
  40.594 116.181
  54.656  55.053  64.632  66.534  67.669  67.767  67.769  67.969  67.978  68.187
   71.23  72.961  73.224  73.961  74.561   74.76  75.301  77.061  77.559  79.063
  79.356  80.374  80.705  81.348  81.353  81.415  81.427  83.409  86.641  87.358
 101.683 102.067
  117.74 117.866 120.905 120.898 120.951 120.955 121.071 121.083 122.069 122.079
  122.22 122.301 122.306 122.322 122.335 122.337 122.318 122.255 122.237 122.175
 122.163 122.085  122.06 122.012 121.006 121.001 120.864 120.494   120.4 120.379
 116.291 116.181
  117.74  40.529  40.436  40.417  40.406   55.42  55.799  86.649   88.14   120.4
 120.591 120.648 120.657  120.66 120.662 120.663 120.665 120.602 120.584  120.53
 120.493 120.363  40.594  40.594  40.594  40.594  40.594  40.594  40.594  40.594
  40.594 116.181
BR Coef=-1 , 0 , 0 ,, 0 ,,,0.8,-1,,0,
WSPro=,,,, 1 ,,,, 0 ,,,, 0 ,,,,-1 ,-1 ,-1 , 0 , 0 , 0 , 0 , 0
BC Mult= 1 ,0,68,0,67
BC Mult= 3 ,68,82,67,82
BC Mult= 1 ,82,400,82,400
BC Design=,, 0 ,, 0 ,,,,,,
BC Use User HTab Curves=0
BC User HTab FreeFlow(D)= 0

Type RM Length L Ch R = 1 ,1231.045,76.511,74.718,72.925
XS GIS Cut Line= 6
  529839.8164404 4779160.7673169  529888.3078166 4779170.2496899
  529917.1535635 4779190.2786732  529969.7485025 4779199.0769225
  530060.6829718 4779226.1387898  530209.9272401        4779265.
#Sta/Elev= 30
       0 126.801  10.645 122.303  11.967 121.912   16.52 121.471  25.693 121.225
  29.312 121.036  49.411 121.134   67.66  120.77  68.172 117.967  70.623 117.595
  76.523 117.514  79.192 117.728  80.185 118.773  80.445   120.8   80.49 120.792
 122.358 120.662 150.198 120.923 161.753 120.668 209.833 121.645247.7024121.6271
255.6877121.9511263.6729121.9789286.6306 121.764287.6288122.5084 326.557123.6561
335.5404124.3216353.5073124.6198360.4944124.5699361.4926124.0734388.4429122.4281
#Mann= 4 ,-1 , 0
       0      .1       0  25.693      .1       0  68.172    .036       0
  80.185      .1       0
Levee=0,,,-1,343.61,124.44,,Levee 42
#XS Ineff= 2 ,-1
   35.46   52.42  126.52   97.36     237  130.04
Permanent Ineff=
       T       T
#Block Obstruct= 4 ,-1
  148.72  207.58  129.28  237.53  245.64  135.24  288.28  328.81  130.28
  361.94  386.26   143.6
Bank Sta=67.66,80.49
XS Rating Curve= 0 ,0
Exp/Cntr=0.5,0.3

Type RM Length L Ch R = 1 ,1156.328,20.618,23.261,25.798
XS GIS Cut Line= 4
  529804.9874122 4779235.0745122  529881.0140122 4779253.9159122
  529923.6638122 4779259.1528122  530220.5046413 4779269.4063003
#Sta/Elev= 30
       0 126.487   3.966 126.262   7.932 125.509  12.889 125.313   40.65 120.154
  51.557 120.141  55.523 119.427  58.497 119.129  62.463 119.632  86.321 119.017
  89.319 118.381  91.318 117.429  92.317 117.265 108.306 116.563 109.305  116.68
 110.304 117.231 112.303 119.198 143.224  119.53 149.204 119.761 150.201  120.03
 178.109 120.649 215.984 120.839 314.657 121.983 327.614 122.289 362.499 124.632
 367.483 124.697  374.46  124.47 385.423 124.517 414.328 122.269 418.315 122.391
#Mann= 3 ,-1 , 0
       0      .1       0  86.321    .036       0 112.303      .1       0
Levee=0,,,-1,365.64,124.68,,Levee 42
#XS Ineff= 2 , 0
           77.44  134.03  119.21           135.6
Permanent Ineff=
       T       T
#Block Obstruct= 6 ,-1
    11.1   38.85  132.53  115.24  141.67   136.3  148.81  161.76   128.5
  230.84  297.36  134.44  328.63  359.91  143.88  388.11  409.69  143.96
Bank Sta=86.321,112.303
XS Rating Curve= 0 ,0
Exp/Cntr=0.3,0.1

Type RM Length L Ch R = 5 ,1155.736,,,
BEGIN DESCRIPTION:
E153
END DESCRIPTION:
IW Pilot Flow=0
#Inline Weir SE= 5
       0       0    78.7  117.77   89.97  117.77  111.46  117.71  122.25  117.71
IW Dist,WD,Coef,Skew,MaxSub,Min_El,Is_Ogee,SpillHt,DesHd
0.1,1.3,1.7,0,0.98,, 0 ,,,0,0,

Type RM Length L Ch R = 1 ,1133.066,8.865,9.319,9.88
XS GIS Cut Line= 5
  529804.8397122 4779241.7007122  529889.3729122 4779268.4929122
  529909.8838122 4779289.6791122  530012.9753924 4779326.0432173
  530222.9383242 4779321.3248688
#Sta/Elev= 30
       0 126.654   5.978 125.546  27.899 123.135  34.873 121.337  37.862 120.496
  67.754 118.463  73.732 118.429  78.714 119.051  96.541 118.853 100.473 118.199
 103.422 115.087 105.387  114.92  106.37 115.274 108.336 118.405 109.319 118.742
 182.762 119.588 225.495 119.618 310.095 121.868 319.053 121.914 320.048 121.488
 402.661 124.148 423.563 124.239 425.553 125.617 426.549 125.478 427.544 129.619
 428.539 136.062 429.535  139.92  430.53 141.811 433.516 142.914 437.497     143
#Mann= 4 ,-1 , 0
       0      .1       0  34.873      .1       0  96.541    .036       0
 108.336      .1       0
#XS Ineff= 2 , 0
           94.71  132.87  111.89          134.08
Permanent Ineff=
       T       T
#Block Obstruct= 8 ,-1
   54.63   63.44  130.58   146.7  160.79  134.24  170.93   181.5  141.08
   197.8  219.38  137.84  228.19  249.78  139.16  262.56  305.73  147.26
  326.43  376.65  146.12  383.26  388.55  138.08
Bank Sta=100.473,108.336
XS Rating Curve= 0 ,0
Exp/Cntr=0.5,0.3

Type RM Length L Ch R = 4 ,1128.406,,,
BEGIN DESCRIPTION:
E154
END DESCRIPTION:
Bridge Culvert--1,0,-1,-1, 0
Deck Dist Width WeirC Skew NumUp NumDn MinLoCord MaxHiCord MaxSubmerge Is_Ogee
0.01,9.12,1.44,0, 32, 32, , , 0.95, 0, ,,,
  84.423  84.985  93.478 100.306 100.318 101.457 101.705 101.711 101.714 101.754
 102.054 102.671 103.288 104.074 104.598 105.337 105.988 106.325 106.912 107.062
 107.506 108.041 108.247 108.453 108.551 108.723 108.733 108.883 110.461 110.746
 123.802 124.102
 116.439 116.608 119.166 119.126 119.823 119.821 119.821 119.821 119.611 119.611
 119.617 119.628 119.639 119.653 119.663 119.676 119.688 119.694 119.704 119.707
 119.697 119.685 119.681 119.676 119.674  119.67 118.696 118.696 118.696 118.696
 115.841 115.775
 116.439  43.049  42.837  42.666  42.666  42.638 115.193 115.223 115.241 115.441
  116.25 117.093 117.585  117.95 118.073 118.108 118.005   117.9 117.619 117.505
 117.169 116.524 116.157 115.622 115.182  77.277  75.153  41.985  41.955   41.95
  41.706 115.775
  81.229  81.791  90.284  97.112  97.124  98.263  98.511  98.517   98.52   98.56
   98.86  99.477 100.094  100.88 101.404 102.143 102.794 103.131 103.718 103.868
 104.312 104.847 105.053 105.259 105.357 105.529 105.539 105.689 107.267 107.552
 120.608 120.908
 116.439 116.608 119.166 119.126 119.823 119.821 119.821 119.821 119.611 119.611
 119.617 119.628 119.639 119.653 119.663 119.676 119.688 119.694 119.704 119.707
 119.697 119.685 119.681 119.676 119.674  119.67 118.696 118.696 118.696 118.696
 115.841 115.775
 116.439  43.049  42.837  42.666  42.666  42.638 115.193 115.223 115.241 115.441
  116.25 117.093 117.585  117.95 118.073 118.108 118.005   117.9 117.619 117.505
 117.169 116.524 116.157 115.622 115.182  77.277  75.153  41.985  41.955   41.95
  41.706 115.775
BR Coef=-1 , 0 , 0 ,, 0 ,,,0.8,0,,0,
WSPro=,,,, 1 ,,,, 0 ,,,, 0 ,,,,-1 ,-1 ,-1 , 0 , 0 , 0 , 0 , 0
BC Mult= 1 ,0,100,0,95
BC Mult= 3 ,100,108,95,106
BC Mult= 1 ,108,500,106,500
BC Design=,, 0 ,, 0 ,,,,,,
BC Use User HTab Curves=0
BC User HTab FreeFlow(D)= 0

Type RM Length L Ch R = 1 ,1123.747,60.837,59.112,57.387
XS GIS Cut Line= 5
  529803.6931122 4779249.3725122  529885.9573122 4779274.7632122
  529901.2370122 4779296.6123122  530013.5071349 4779335.5038908
  530231.8618281 4779335.9269662
#Sta/Elev= 30
       0 126.502  17.812 123.954  25.729 123.485  39.583 120.165  84.114 118.162
  89.056 118.259  95.968 117.623  97.943 114.472  99.918 113.866 102.881 113.623
 104.855 114.446 105.843 118.021 107.818 118.937 124.737 118.473  167.67 119.317
 232.567  119.44 257.494 120.291 266.467 120.221 273.447 121.307 278.432 120.744
 310.338   121.1 311.335 120.896 361.189  122.18 376.145 122.836 390.104 122.897
 414.034 123.919 426.996 123.858 430.984 122.647 436.966 121.684 449.928 121.439
#Mann= 3 ,-1 , 0
       0      .1       0  95.968    .036       0 105.843      .1       0
Levee=0,,,-1,414.98,123.97,,Levee 43
#XS Ineff= 3 ,-1
     3.3   95.15   134.8   95.82   98.52     119  107.49  452.86  136.64
Permanent Ineff=
       T       T       T
#Block Obstruct= 8 ,-1
    51.1   81.94  132.44   88.55   95.59   125.9  107.93  118.06   133.4
   134.8  166.52  134.48  186.34  223.79   138.2   234.8  258.15  138.68
   285.9   351.1  145.34  392.95  412.78  144.56
Bank Sta=95.968,105.843
XS Rating Curve= 0 ,0
Exp/Cntr=0.5,0.3

Type RM Length L Ch R = 1 ,1064.635,4.091,4.093,4.095
XS GIS Cut Line= 5
  529786.9675122 4779309.0818122  529840.0195122 4779321.3245122
  529863.3667122 4779333.9245122  529977.9636353 4779372.8920086
   530236.146124 4779362.6721272
#Sta/Elev= 30
       0 126.154  13.859 125.058  19.799 123.778  43.557 121.754  45.537 119.868
  46.527 119.442  56.412 119.174  59.359 117.377  60.342 117.012   63.29 114.324
   67.22 113.803  70.168 113.975  72.133   114.6  73.116 115.233  74.098 117.341
 145.466 118.968 193.088     119 224.963 119.568 251.899  118.89 295.794  120.27
 335.699 120.519 378.596 119.978  385.58  120.38 400.544  119.91 429.475 123.192
 445.437 123.145 446.435 122.976 449.427 120.749 450.425 120.613 460.401 121.339
#Mann= 3 ,-1 , 0
       0      .1       0  59.359    .036       0  74.098      .1       0
Levee=0,,,-1,441.41,123.17,,Levee 43
#XS Ineff= 2 ,-1
     .22   29.07     135   75.77  462.33  137.72
Permanent Ineff=
       T       T
#Block Obstruct= 8 ,-1
   75.33   92.95  131.92   99.56  137.89  133.89  146.26  188.99  133.41
  196.48  222.03  135.92  229.07  247.14  137.15   253.3  262.11  132.35
  298.24  371.81  139.71  413.66  427.75   145.2
Bank Sta=59.359,74.098
XS Rating Curve= 0 ,0
Exp/Cntr=0.3,0.1

Type RM Length L Ch R = 1 ,1060.542,32.59,30.154,27.718
XS GIS Cut Line= 5
  529788.9732122 4779314.8003122  529842.0252122 4779327.0430122
  529865.3724122 4779339.6429122  529973.7069699 4779376.4810395
  530234.3208619 4779366.9310723
#Sta/Elev= 30
       0 125.591   7.919  125.21  41.577 121.644  44.547 119.394  53.456 119.254
  54.446 118.682  55.429 117.602  56.411 116.411  57.394 114.985  58.377 114.264
  62.307 113.798   67.22 114.511  70.168 116.474   70.48  117.93  95.902  117.87
 144.657 119.024 254.355 118.835 275.338  119.87 325.296 120.411 326.296 120.711
 337.287 120.283 360.268 120.789 374.256  119.92 399.235 119.836 403.232 119.982
 428.212 122.963   442.2 123.157 444.198 122.976 449.194 120.597 456.189 121.028
#Mann= 3 ,-1 , 0
       0      .1       0  55.429    .036       0   70.48      .1       0
Levee=0,,,-1,437.44,122.97,,Levee 43
#XS Ineff= 2 ,-1
     .44   18.28  133.68   72.91  457.93134.7534
Permanent Ineff=
       T       T
#Block Obstruct= 9 ,-1
   73.13   92.07  133.19   98.24  138.77  133.52  147.58  189.43  133.99
  197.36  241.85  136.55  260.35  274.45  131.37  286.78  321.59  144.02
  325.11  333.48  143.97  341.41  359.03  139.31  409.69  426.87  143.04
Bank Sta=56.411,70.168
XS Rating Curve= 0 ,0
Exp/Cntr=0.3,0.1

Type RM Length L Ch R = 1 ,1030.388,65.548,64.859,64.168
XS GIS Cut Line= 5
  529722.3136967 4779359.2708863  529800.8957832 4779369.5750236
  529873.7799122 4779357.3109122  529976.0082381  4779380.677578
  530235.5377033 4779369.9731759
#Sta/Elev= 30
       0 135.373    .991 134.225   1.981 128.633   2.972 126.911   5.944 126.419
   57.46 124.637  59.441 123.321   72.32 123.083  79.255 121.084  85.247 120.416
  88.244 122.487  93.237 122.599 102.226 119.114 119.205 118.817 121.834 117.833
 122.202 117.512 125.198 113.819 129.193 115.268 133.188 114.459  133.74  117.42
  134.27   118.4 311.978 118.816 312.977 119.847 373.919 120.546 461.836 119.825
 471.826 121.687 503.796 123.077 505.794 122.827  509.79 120.659 517.783 121.075
#Mann= 3 ,-1 , 0
       0      .1       0 121.834    .036       0  133.74      .1       0
Levee=0,,,-1,499.56,122.79,,Levee 43
#XS Ineff= 2 , 0
            90.4  131.05  136.92          131.19
Permanent Ineff=
       T       T
#Block Obstruct= 9 ,-1
   13.74   28.02  134.73   45.46   57.62  132.21  136.39  157.53  130.44
  163.35  201.41  133.01  212.51  249.52  135.71  256.39  294.45  137.11
  314.54  336.74  132.35  346.26  381.67  138.89  472.07  487.93  142.01
Bank Sta=122.202,133.74
XS Rating Curve= 0 ,0
Exp/Cntr=0.5,0.3

Type RM Length L Ch R = 1 ,965.5293,6.065,6.066,6.068
XS GIS Cut Line= 6
  529660.2547828 4779424.3719039  529783.1769809 4779447.5707518
  529847.0067122 4779430.4019122  529892.2405122 4779413.6676122
  529966.7043794 4779394.6571931  530237.9713862  4779374.232121
#Sta/Elev= 30
       0 125.577  11.914 125.025  21.841 125.653  55.597 122.483  79.424 122.377
  98.287 120.824 123.107 120.399 126.079 118.857 133.971 120.312 174.419 117.711
 200.201 117.406 203.002 114.372 205.955 113.455 207.923  114.11 208.908 115.321
 209.892 117.901 326.237 118.854 329.226 120.155 379.049 119.652 380.046 118.591
 381.042 118.581 436.844 120.429 459.763 119.624  474.71 120.299 531.508 119.844
 559.409 122.715  570.37 122.862 575.352 122.559 580.334 120.605 588.306 121.219
#Mann= 3 ,-1 , 0
       0      .1       0 200.201    .036       0 209.892      .1       0
Levee=0,,,-1,565.64,122.6,,Levee 43
#XS Ineff= 2 , 0
          172.33  131.47  212.51          134.13
Permanent Ineff=
       T       T
#Block Obstruct= 9 ,-1
   63.44    79.3  132.07  139.56  172.33  130.86  211.98  235.24  133.85
  242.11  261.67  133.01  285.99  305.02  132.77  329.87  377.97  134.73
  384.85  407.05  137.72  418.15  435.07   133.1  543.96  558.24  143.13
Bank Sta=200.201,209.892
XS Rating Curve= 0 ,0
Exp/Cntr=0.5,0.3

Type RM Length L Ch R = 4 ,962.5384,,,
BEGIN DESCRIPTION:
E155
END DESCRIPTION:
Bridge Culvert--1,0,-1,-1, 0
Deck Dist Width WeirC Skew NumUp NumDn MinLoCord MaxHiCord MaxSubmerge Is_Ogee
0.01,5.87,1.44,0, 29, 29, , , 0.95, 0, ,,,
     190 190.177 197.294 198.314 200.661 200.674 200.915 200.918 201.311 201.675
 202.076 202.748 203.393 204.642 204.733 205.338 205.446 206.191 207.084 207.175
 208.206 209.157 209.631 209.899 210.088 210.123 210.591 222.808 222.875
 116.024 116.092 117.709 117.819 117.818 118.711 118.712 118.527 118.599 118.664
 118.737 118.859 118.976 119.202  119.21 119.263 119.257 119.218 119.171 119.166
   119.1  119.04 119.009 118.992  118.98 118.978 118.948 115.931 115.915
 116.024  67.094  67.035  67.026  67.006  67.006  67.004  67.004  67.001 115.504
 115.995 116.596 117.001 117.438  117.47 117.541 117.554 117.531 117.349 117.309
 116.849 116.098 115.538 115.127  67.016  67.016  67.006  66.752 115.915
 194.818 195.118 202.235 203.255 205.602 205.615 205.856 205.859 206.252 206.616
 207.017 207.689 208.334 209.583 209.674 210.279 210.387 211.132 212.025 212.116
 213.147 214.098 214.572  214.84 215.029 215.064 215.532 227.749 227.816
 116.024 116.092 117.709 117.819 117.818 118.711 118.712 118.527 118.599 118.664
 118.737 118.859 118.976 119.202  119.21 119.263 119.257 119.218 119.171 119.166
   119.1  119.04 119.009 118.992  118.98 118.978 118.948 115.931 115.915
 116.024  67.094  67.035  67.026  67.006  67.006  67.004  67.004  67.001 115.504
 115.995 116.596 117.001 117.438  117.47 117.541 117.554 117.531 117.349 117.309
 116.849 116.098 115.538 115.127  67.016  67.016  67.006  66.752 115.915
BR Coef=-1 , 0 , 0 ,, 0 ,,,0.8,-1,,0,
WSPro=,,,, 1 ,,,, 0 ,,,, 0 ,,,,-1 ,-1 ,-1 , 0 , 0 , 0 , 0 , 0
BC Mult= 1 ,0,200,0,205
BC Mult= 3 ,200,216,205,216
BC Mult= 1 ,216,600,216,600
BC Design=,, 0 ,, 0 ,,,,,,
BC Use User HTab Curves=0
BC User HTab FreeFlow(D)= 0

Type RM Length L Ch R = 1 ,959.4634,44.48,44.499,44.518
XS GIS Cut Line= 6
  529657.2126792 4779434.1066354  529780.0247007 4779455.0776081
  529849.0124122 4779436.1203122  529894.2462122 4779419.3860122
  529969.1400169 4779400.2658312  530236.5644133 4779376.9826897
#Sta/Elev= 30
       0 125.281  11.961 124.375  20.931 125.202  33.888  123.55  48.839 123.782
  49.836 122.799  55.816 122.064  68.773 121.958  92.695 119.504  95.685 120.638
 102.662 120.839 106.649 119.948 120.603 118.497 204.586 117.549 205.978 116.589
 207.946 114.339 210.899 113.589 212.868 114.222 214.836  116.45  215.68  118.07
 259.229 118.366 261.211 119.036 384.528   118.5 415.462 119.603 533.214 119.657
  564.15 122.636 572.133 122.724 579.119 122.511 584.109 120.528 590.096 121.002
#Mann= 3 ,-1 , 0
       0      .1       0 204.586    .036       0  215.68      .1       0
Levee=0,,,-1,573.04,122.74,,Levee 43
#XS Ineff= 2 , 0
          100.97  133.29  216.74          131.28
Permanent Ineff=
       T       T
#Block Obstruct= 9 ,-1
   36.48   49.16   132.4   74.01   90.93  132.13  216.22   243.7  127.51
  260.62  284.93  132.03  291.28  327.22  135.92  333.04   382.2  131.44
  388.02  411.81  137.79  423.44  453.04  142.64  547.14  562.47  144.77
Bank Sta=205.978,214.836
XS Rating Curve= 0 ,0
Exp/Cntr=0.5,0.3

Type RM Length L Ch R = 1 ,914.9646,21.482,20.987,20.492
XS GIS Cut Line= 4
  529649.3708121 4779454.0831159  529845.6079122 4779484.6141122
  529932.5204122 4779452.9652122  530228.0465231  4779387.325842
#Sta/Elev= 30
       0 138.073   2.994  136.55   3.992  128.73    4.99 125.465   5.988 124.624
    9.98 124.418  15.968 122.858  29.939 121.805  46.905 121.556  55.887 120.423
  65.867 121.751  76.844 119.524   93.81 119.091 102.792 117.522 186.622  117.83
 224.457 116.949 227.441 114.797  229.43 114.618 237.387 115.264  238.94  117.05
 378.017 118.549 402.995 117.905 431.969 119.208 474.931 119.888  498.91  119.32
 551.862 119.406 560.854 120.342 561.853 121.177 578.837 122.429 593.823 122.104
#Mann= 3 ,-1 , 0
       0      .1       0 224.457    .036       0  238.94      .1       0
Levee=0,,,-1,586.78,122.51,,Levee 43
#XS Ineff= 2 , 0
          207.75  132.73  241.59          132.77
Permanent Ineff=
       T       T
#Block Obstruct= 12 ,-1
   35.95   48.63  130.63  124.23   145.9  130.35  152.25  164.93  131.33
  190.84  208.28  131.98  241.59  261.67  131.75  269.07  303.96  132.96
  311.37  346.78  135.62  352.07  374.27  137.58   378.5  399.65  128.62
  403.35  430.84  132.49  440.35  468.37  128.15  562.47  577.27  143.32
Bank Sta=224.457,238.94
XS Rating Curve= 0 ,0
Exp/Cntr=0.3,0.1

Type RM Length L Ch R = 1 ,893.9775,28.072,28.243,28.414
XS GIS Cut Line= 4
  529627.7380752 4779477.8791264  529854.1578122 4779508.5986122
  529938.8780122 4779464.0989122  530228.6549439 4779393.4100492
#Sta/Elev= 30
       0 122.244  86.808 118.899 110.755 119.241 117.739 118.718 120.733 117.488
 122.728 117.228  130.71  117.51 178.604 116.887  198.56 117.357  256.56  116.63
  256.57 115.257 257.402 114.527 258.399 114.455  267.37 114.868 268.367 115.131
 269.364 116.734 269.463 117.055  377.06  118.17 400.004 117.542 404.992 118.214
 424.943 118.254 430.928 117.771 431.926   118.2 464.845 119.102 496.767 119.472
 583.555 119.323 588.542 120.256 591.535 121.839 621.462 122.513 622.459 125.053
#Mann= 3 ,-1 , 0
       0      .1       0  256.56    .036       0 269.463      .1       0
#XS Ineff= 2 , 0
          255.33  135.76  271.98          135.06
Permanent Ineff=
       T       T
#Block Obstruct= 12 ,-1
   94.98  111.01  134.31   158.5  187.49  129.93  202.91  238.06  124.47
  246.08  255.33  135.29  271.37  292.33  134.64  299.12  334.89  130.67
  341.67  376.21  137.07  380.53  400.26  130.67  406.43  417.53  127.59
  432.95  461.32  134.64  469.34  485.37  132.31  591.45  608.11  143.79
Bank Sta=256.56,269.364
XS Rating Curve= 0 ,0
Exp/Cntr=0.3,0.1

Type RM Length L Ch R = 5 ,892.4471,,,
BEGIN DESCRIPTION:
E156
END DESCRIPTION:
IW Pilot Flow=0
#Inline Weir SE= 5
       0       0   97.57  114.75  124.02  114.75  139.14  114.81  192.75  114.81
IW Dist,WD,Coef,Skew,MaxSub,Min_El,Is_Ogee,SpillHt,DesHd
1.8,1.8,1.7,0,0.98,, 0 ,,,0,0,

Type RM Length L Ch R = 1 ,865.7347,39.621,39.849,40.076
XS GIS Cut Line= 4
  529618.0033436 4779503.8384107  529859.0827122 4779535.7021122
  529978.1365122 4779480.0083122  530238.9980962 4779398.8858357
#Sta/Elev= 30
       0 128.019    .997 124.678   1.993  126.63   3.986 121.926   76.74 119.664
  89.696 118.587 140.524 118.529 142.517  117.66  156.47 117.398   276.3  116.16
 276.867 114.711 277.031 112.276 278.027 111.461  282.01 111.248 285.993 112.318
  286.78  114.76  288.02  116.16 306.903  115.74 315.865 116.918 420.475 118.012
 446.397  117.52 504.224 119.164 595.949  119.35 603.925 119.863 607.913 122.184
  638.82 122.448 639.817 125.358 641.811 140.912 642.808 143.382 647.793 144.567
#Mann= 3 ,-1 , 0
       0      .1       0 276.867    .036       0  286.78      .1       0
#XS Ineff= 2 , 0
          275.68  136.65  288.63          129.09
Permanent Ineff=
       T       T
#Block Obstruct= 12 ,-1
    4.32   37.62   128.9   49.34   64.76  143.65  122.11  141.23  121.39
  263.96  275.68  136.09  288.63  299.74  128.67  316.39  351.54  132.59
  358.33  392.86  132.31   397.8  418.77  135.62  424.32  444.67  130.72
  447.75  479.21  130.25  484.76   519.3  127.55  608.11  624.14  144.07
Bank Sta=276.867,286.78
XS Rating Curve= 0 ,0
Exp/Cntr=0.5,0.3

Type RM Length L Ch R = 1 ,825.8861,10.672,10.669,10.666
XS GIS Cut Line= 5
  529618.0033436 4779531.9609686  529863.5447122 4779574.2140122
  529998.4313122 4779521.0226122  530250.5580899 4779428.6984512
530302.9958227094779409.49672368
#Sta/Elev= 30
       0 119.925  16.942 119.853  31.891 118.784  50.827 118.714  53.816 118.089
  72.752  118.13   96.67 117.446 198.324 117.661  199.32 116.986   205.3 115.995
  208.29 115.982 209.286 117.137  265.15 116.546  266.15 115.573 280.149 115.635
 281.149 115.964  294.19  115.76 295.149 111.394 297.149 110.912 298.149 111.014
 300.148 112.255 301.148 115.935 333.147 116.649 447.047 117.133 502.943 118.652
671.5812118.9409 674.575119.4485683.5562119.4613699.5226120.2497718.4828122.2126
#Mann= 3 ,-1 , 0
       0      .1       0  294.19    .036       0 301.148      .1       0
#XS Ineff= 3 ,-1
       0  264.32  136.08  278.41  291.81  135.17  303.79718.4828  133.73
Permanent Ineff=
       T       F       T
#Block Obstruct= 10 ,-1
   51.19   74.01  146.48  107.93  197.97  133.25  211.54   265.2  135.28
  279.38  292.33  135.23  302.82  323.79  132.56  334.27  399.65  139.17
  423.08  443.44  135.92  450.84  491.54  136.67  507.58  535.33  134.05
  605.02  621.06  122.59
Bank Sta=294.19,301.148
XS Rating Curve= 0 ,0
Exp/Cntr=0.5,0.3

Type RM Length L Ch R = 4 ,820.4001,,,
BEGIN DESCRIPTION:
E157
END DESCRIPTION:
Bridge Culvert--1,0,-1,-1, 0
Deck Dist Width WeirC Skew NumUp NumDn MinLoCord MaxHiCord MaxSubmerge Is_Ogee
0.01,10.47,1.44,0, 30, 30, , , 0.95, 0, ,,,
 280.924 281.074 290.398 293.888   293.9 294.141 294.288 294.319 294.589 295.215
 295.788 296.679 297.312 297.505 297.866 298.567  298.85 299.368 300.028  300.53
  300.82 300.887 300.893   300.9 300.925 300.949 301.496 305.833 314.989  315.31
 112.742 112.788  115.64 115.662 116.764 116.771 116.775 116.775 116.783   116.8
 116.815 116.839 116.856 116.861 116.871  116.89 116.898 116.912  116.93 116.943
 116.951 116.953 115.798 115.799 115.799 115.799 115.805  115.85 113.214 113.121
 112.742  39.765  40.022  40.118  40.119  40.125 111.793  112.07 112.962 113.875
 114.349 114.761 114.882 114.894 114.887 114.759 114.661 114.401 113.869 113.192
 112.505 112.229 112.203 112.173 111.985 111.793  40.049  40.096  40.196 113.121
 289.324 289.474 298.798 302.288   302.3 302.541 302.688 302.719 302.989 303.615
 304.188 305.079 305.712 305.905 306.266 306.967  307.25 307.768 308.428  308.93
  309.22 309.287 309.293   309.3 309.325 309.349 309.896 314.233 323.389  323.71
 112.742 112.788  115.64 115.662 116.764 116.771 116.775 116.775 116.783   116.8
 116.815 116.839 116.856 116.861 116.871  116.89 116.898 116.912  116.93 116.943
 116.951 116.953 115.798 115.799 115.799 115.799 115.805  115.85 113.214 113.121
 112.742  39.765  40.022  40.118  40.119  40.125 111.793  112.07 112.962 113.875
 114.349 114.761 114.882 114.894 114.887 114.759 114.661 114.401 113.869 113.192
 112.505 112.229 112.203 112.173 111.985 111.793  40.049  40.096  40.196 113.121
BR Coef=-1 , 0 , 0 ,, 0 ,,,0.8,0,,0,
WSPro=,,,, 1 ,,,, 0 ,,,, 0 ,,,,-1 ,-1 ,-1 , 0 , 0 , 0 , 0 , 0
BC Mult= 1 ,0,294,0,303
BC Mult= 3 ,294,301,303,310
BC Mult= 1 ,301,800,310,700
BC Design=,, 0 ,, 0 ,,,,,,
BC Use User HTab Curves=0
BC User HTab FreeFlow(D)= 0

Type RM Length L Ch R = 1 ,815.2168,31.55,31.932,32.314
XS GIS Cut Line= 4
  529612.5951594 4779546.0222476  529864.7373122 4779585.2556122
  530002.5944122 4779530.7679122  530237.7812547 4779442.6921279
#Sta/Elev= 30
       0 131.904   1.994 131.876    2.99 131.142   3.987 118.983   4.984 118.905
  53.826 118.673   58.81 118.596    61.8 118.071  67.781 118.211 105.659  117.08
 250.192 115.708 257.166 115.377  303.55  115.65  304.17  112.88  304.32  111.27
 304.919 110.892  307.15  111.01  307.75  111.38  308.57  115.84 325.812 116.275
 326.807 116.614 327.802 117.747 410.388 117.536 438.292 116.912 504.067 118.111
 505.063 118.901 557.882 118.595 623.657 118.943 635.616 118.747 654.551 118.971
#Mann= 3 ,-1 , 0
       0      .1       0  303.55    .036       0  308.57      .1       0
#XS Ineff= 3 ,-1
       0  271.37   137.4     280   302.2  128.27  308.99 654.551  130.33
Permanent Ineff=
       T       F       T
#Block Obstruct= 9 ,-1
   65.37   95.59  145.33  117.18  246.08  140.53   257.8  271.37   137.4
  280.62  302.82  128.07  308.99  321.94  129.67  329.96  407.67  150.53
   412.6  429.87  133.33  455.77  500.18     135  506.34   545.2  132.47
Bank Sta=303.55,308.57
XS Rating Curve= 0 ,0
Exp/Cntr=0.5,0.3

Type RM Length L Ch R = 1 ,783.2848,55.975,55.97,55.965
XS GIS Cut Line= 4
529565.4379493024779556.04010312529874.3157043154779610.18368492
530065.5831284014779556.76071474530315.5498653964779489.48734489
#Sta/Elev= 30
       0 121.152    4.16 119.592  40.242 118.611  90.695  118.49  97.669 117.774
 114.976 117.831 117.991 117.016 122.909 116.808 286.884 115.794 319.843 114.669
  358.13  115.55 358.706 112.206  358.79  110.99 361.719  110.15 364.466  110.99
  365.09   115.6 384.211 115.486 386.233  116.42 479.934  117.21  596.92 117.367
 666.812 118.325 672.673 118.301 672.886 117.755 684.295 117.915 750.109 117.658
 762.116 118.856 762.932 119.722 764.017 122.281 764.564 121.806 771.037 121.891
#Mann= 4 ,-1 , 0
       0      .1       0 358.706    .036       0 364.466      .1       0
 684.295    .045       0
#XS Ineff= 3 ,-1
       0  300.97  139.17  329.16  350.31  138.19  364.41 771.037  134.03
Permanent Ineff=
       T       F       T
#Block Obstruct= 9 ,-1
   40.88   59.21  132.63  171.28  226.96  140.05  328.46  350.31  138.09
  365.11   377.8  129.46  391.19  462.38  135.67   479.3  536.39   136.6
  598.41  643.52   128.9  662.56  672.42  121.71  693.57  700.62  121.48
Bank Sta=358.13,365.09
XS Rating Curve= 0 ,0
Exp/Cntr=0.3,0.1

Type RM Length L Ch R = 1 ,727.3147,49.507,50.74,51.972
XS GIS Cut Line= 4
529391.3593944674779597.93329951529874.4377944674779668.28449951
530052.6609944674779618.25699951530345.0094944674779536.96219951
#Sta/Elev= 30
       0 135.108   5.469 133.775   7.163 130.745    7.49  129.43   8.501 117.308
   9.511 116.476   95.12 117.575 277.414 115.962 348.577 115.073 349.056 113.101
 389.478 112.728 391.341 114.405 403.876 114.234 417.773 115.351  475.94 114.919
  485.83 113.861 545.207  114.06 545.407  110.92 547.702 110.652 553.955 110.901
 554.593 111.307 554.658 114.168 571.959 115.022 722.183 116.991  839.82 117.505
  871.22 116.614 926.658 117.954 935.666 116.899 962.987 116.976 976.727 117.875
#Mann= 4 ,-1 , 0
       0      .1       0 389.478      .1       0 545.207    .036       0
 554.658      .1       0
Levee=-1,110.13,117.05,0,,,Levee 4,
#XS Ineff= 3 ,-1
       0  478.41  139.91  499.56  541.85  139.63  556.83 976.727  135.25
Permanent Ineff=
       T       F       T
#Block Obstruct= 10 ,-1
   45.81  109.25   142.4  165.64  238.77   140.6  313.66  347.14  142.47
   497.8  541.85  139.73  556.83  649.35  127.93  662.56  689.87   127.2
  726.87  785.02  133.33  802.64  837.89  132.73  893.39  925.11  130.13
  939.21  963.88  132.13
Bank Sta=545.207,554.658
XS Rating Curve= 0 ,0
Exp/Cntr=0.5,0.3

Type RM Length L Ch R = 1 ,676.5748,23.383,23.718,24.053
XS GIS Cut Line= 4
529380.415825951   4779641.70739529881.3778165774779697.60067324
530039.5064696534779706.24968232530357.5163321374779558.84926707
#Sta/Elev= 30
       0 114.951 109.791 116.229 272.033 115.915 298.799 114.283 310.998 112.007
 375.357 110.961 377.623  113.86 380.449 114.704 408.685 114.269 443.088 115.147
 481.323 114.614 485.348 113.676 495.887 113.412  562.79 113.886 562.937  110.93
 565.886  110.51 573.023 110.725  574.16  113.74 587.589 114.507 645.338 114.063
 648.398 114.604 746.896 115.964 794.783 116.114 804.912 116.797 837.635 115.773
 848.174 116.518 881.499 115.963 947.773 116.986 971.775 116.3591012.946 118.183
#Mann= 4 ,-1 , 0
       0      .1       0 375.357      .1       0  562.79    .036       0
  574.16      .1       0
Levee=-1,174.45,116.21,0,,,Levee 4,
#XS Ineff= 3 ,-1
    1.06  481.06  143.04  505.37  548.72  128.71  577.271012.946  133.29
Permanent Ineff=
       F       T       T
#Block Obstruct= 9 ,-1
      37  117.36  142.32  185.02  273.83  141.52  383.79  413.39  121.76
  505.37  548.72   128.8  576.21  652.33  130.96  679.82  762.29  132.32
  802.47   836.3  129.92   851.1   865.9  136.48  905.02   945.2  136.64
Bank Sta=562.79,574.16
XS Rating Curve= 0 ,0
Exp/Cntr=0.5,0.3

Type RM Length L Ch R = 4 ,664.2988,,,
BEGIN DESCRIPTION:
E158
END DESCRIPTION:
Bridge Culvert--1,0,-1,-1, 0
Deck Dist Width WeirC Skew NumUp NumDn MinLoCord MaxHiCord MaxSubmerge Is_Ogee
0.01,23.52,1.44,0, 21, 17, , , 0.95, 0, ,,,
 553.822 554.099 560.881 562.627 562.933 562.943  564.12 565.634 567.299 568.567
 569.972 571.199 572.806 573.362 573.393 574.535 574.835 574.971 577.777 586.853
 587.008
 112.678 112.723 113.833 113.848 113.851  115.15 115.145  115.14 115.134 115.129
 115.124  115.12 115.114 115.112 114.013 114.013 114.013 114.013 114.013 111.974
  111.94
 112.678  37.372  37.372  37.372 112.209 112.211 112.448 112.673 112.819  112.86
 112.835 112.753 112.558 112.454 112.449 112.236 112.168  36.788  36.768  36.701
  111.94
   564.5 565.815 565.978 566.168 566.661 567.112 574.466 574.503 577.242 577.256
 579.303 580.174 580.634 580.651  585.53 585.612  587.86
     130     130     130     130     130     130     130     130     130     130
     130     130     130     130     130     130     130
  -28.47  -28.47  -28.47  -28.47  -28.47 113.071 113.075 113.075 113.077 113.077
 113.078 -30.062 -30.067 -30.067 -30.113 -30.114 -30.135
BR Coef=-1 , 0 , 0 ,, 0 ,,,0.8,-1,,0,
WSPro=,,,, 1 ,,,, 0 ,,,, 0 ,,,,-1 ,-1 ,-1 , 0 , 0 , 0 , 0 , 0
BC Mult= 1 ,0,562.9,0,566.65
BC Mult= 3 ,562.9,575,566.65,585.37
BC Mult= 1 ,575,1100,585.37,1100
BC Design=,, 0 ,, 0 ,,,,,,
BC Use User HTab Curves=0
BC User HTab FreeFlow(D)= 0

Type RM Length L Ch R = 1 ,652.8569,37.639,37.704,37.769
XS GIS Cut Line= 4
529381.224641459 4779665.8273895529881.5290547374779714.72399602
530041.3255457834779736.71134618530358.3251476454779582.96926657
#Sta/Elev= 30
       0  139.61   7.498 138.594   8.587 136.692   9.724 130.621  10.596 128.622
  11.601 131.245  12.606 131.085  13.065 129.295  14.059  127.95  14.615 130.223
  14.974 129.499  16.406  119.28  18.633 114.732 102.844 116.709 202.378 116.875
 272.461  111.84 340.824 112.532 347.626 114.611  566.65  113.72 567.107 110.906
 568.545 110.685 578.681  110.87 584.173 113.359 585.368     114 651.471 113.487
 660.128 114.644 807.857 116.473 840.655 115.585 933.445 117.0931016.305 116.665
#Mann= 3 ,-1 , 0
       0      .1       0  566.65    .036       0 584.173      .1       0
Levee=-1,213.57,116.16,0,,,Levee 4,
#XS Ineff= 4 ,-1
    3.17  485.29  143.74  504.32  565.64  133.43   579.3  584.17   113.4
  594.18 1000.18  138.64
Permanent Ineff=
       T       F       T       T
#Block Obstruct= 11 ,-1
  105.73  139.56   140.8  146.96  204.05   141.6  349.96  375.33  127.76
  418.68  486.35129.8867  504.32   566.7  133.44  667.14  685.11  127.84
  725.29  746.43  133.44  807.75  839.47  129.68   851.1  881.76     138
  900.79  919.82  133.92  936.74  986.43  136.88
Bank Sta=566.65,585.368
XS Rating Curve= 0 ,0
Exp/Cntr=0.5,0.3

Type RM Length L Ch R = 1 ,615.1526,4.457,4.421,4.385
XS GIS Cut Line= 4
529363.5119871944779697.79295905529897.0812245524779752.02393555
530046.0695370654779773.55460023 530337.485771764779616.49819694
#Sta/Elev= 30
       0 133.078     .26 137.493   7.296 138.978   8.291 135.719   9.307 124.002
  10.415 114.434  18.277 114.642  20.363  116.45 194.975 115.542  197.27 114.843
 199.321 112.525 293.765 111.034 296.633  113.33 349.138 113.995 366.889 112.205
 401.543 113.775  586.55   112.8 590.261 110.775 600.628 110.204 613.805 112.801
 689.923 113.074 697.892 114.676 781.524 115.443 954.364 116.367 956.472 114.832
 962.643 116.782  977.55 116.568 983.873  114.78 988.089 116.4511017.899 116.377
#Mann= 3 ,-1 , 0
       0      .1       0  586.55    .036       0 613.805      .1       0
Levee=-1,194.54,115.46,0,,,Levee 4,
#XS Ineff= 2 ,-1
    4.23  570.93  135.22  629.08 1032.95  135.52
Permanent Ineff=
       T       T
#Block Obstruct= 8 ,-1
   24.32    79.3  140.26  112.07  178.68  119.08  419.74  464.14  131.74
  779.21   799.3  137.38  832.07   858.5  128.92  875.42  906.08  136.66
  917.71  946.26  135.64   989.6 1004.41  134.02
Bank Sta=586.55,613.805
XS Rating Curve= 0 ,0
Exp/Cntr=0.5,0.3

Type RM Length L Ch R = 4 ,612.9378,,,
BEGIN DESCRIPTION:
E159
END DESCRIPTION:
Bridge Culvert--1,0,-1,-1, 0
Deck Dist Width WeirC Skew NumUp NumDn MinLoCord MaxHiCord MaxSubmerge Is_Ogee
0.01,4.22,1.44,0, 14, 14, , , 0.95, 0, ,,,
 569.781 570.183 580.948 584.067 584.278 584.279 584.283  609.45 609.529 610.273
 610.293 613.709  624.97 625.157
 109.385 109.524 113.261 113.261 113.261 113.552 115.311 115.441 115.441 115.445
 113.261 113.263 109.867 109.811
 109.385   7.614   7.614   7.614 111.783 112.099 112.099 112.229   7.913   7.919
   7.919   7.944   8.025 109.811
 571.939 572.341 583.106 586.225 586.436 586.437 586.441 611.608 611.687 612.431
 612.451 615.867 627.128 627.315
 109.385 109.524 113.261 113.261 113.261 113.552 115.311 115.441 115.441 115.445
 113.261 113.263 109.867 109.811
 109.385   7.614   7.614   7.614 111.783 112.099 112.099 112.229   7.913   7.919
   7.919   7.944   8.025 109.811
BR Coef=-1 , 0 , 0 ,, 0 ,,,0.8,-1,,0,
WSPro=,,,, 1 ,,,, 0 ,,,, 0 ,,,,-1 ,-1 ,-1 , 0 , 0 , 0 , 0 , 0
BC Mult= 1 ,0,584,0,586
BC Mult= 3 ,584,609.5,586,612
BC Mult= 1 ,609.5,1100,612,1100
BC Design=,, 0 ,, 0 ,,,,,,
BC Use User HTab Curves=0
BC User HTab FreeFlow(D)= 0

Type RM Length L Ch R = 1 ,610.7316,0.109,0.109,0.109
XS GIS Cut Line= 4
 529363.219336214779701.61106935529896.702100321 4779756.5673175
530045.7241584914779776.85472287530337.1931207764779620.31630723
#Sta/Elev= 30
       0 126.692    .585  135.27    1.56 138.137   4.808 140.404    8.19 140.538
  62.883  115.32  93.607 115.671 107.056 114.051 112.659  115.66 197.178 115.525
 199.603 114.219   203.1 110.261 279.505  110.58 299.825 113.639 338.654 113.974
  357.87 112.152 402.526  113.77  583.81  112.98 587.171 112.743 591.462 110.761
 604.889 108.667 609.548 111.625 613.793 112.752 782.161 115.419 960.316 114.658
  966.47 116.686 972.635 116.963 985.288 113.855 996.639 116.657 1017.55 116.212
#Mann= 3 ,-1 , 0
       0      .1       0 587.171    .036       0 613.793      .1       0
#XS Ineff= 2 ,-1
   11.63  560.35  137.14  643.88 1018.15  137.26
Permanent Ineff=
       T       T
#Block Obstruct= 8 ,-1
    4.23   61.32  140.98  112.07   138.5  118.78  300.26  306.61  117.88
  414.45  486.34  130.96  774.98  805.64   137.2  834.18  864.85  128.86
   873.3  901.85   135.7  920.88  957.89  136.18
Bank Sta=583.81,613.793
XS Rating Curve= 0 ,0
Exp/Cntr=0.5,0.3

Type RM Length L Ch R = 1 ,610.6224,71.387,72.224,73.061
XS GIS Cut Line= 4
529363.2069387974779701.71016927529896.6897029074779756.66641742
530045.7117610784779776.95382279530337.1807233624779620.41540716
#Sta/Elev= 30
       0 126.043     .71 135.556   1.572 138.092   4.874 140.422   8.155 140.531
  62.895 115.318  93.731 115.647 107.128 114.053 112.784 115.767 197.243 115.525
 202.181 111.235 280.096 111.056 293.012 113.231 338.465 113.973 354.218 112.235
 488.233 114.128 582.549  113.07 587.214  112.74 591.496  110.76  607.07110.5906
 617.299 113.088 693.437  113.25 782.242 115.702 957.893  116.16 960.007 114.696
 962.431 116.256 978.603   116.2   985.3 113.855 996.651  116.641017.549 116.207
#Mann= 3 ,-1 , 0
       0      .1       0 587.214    .036       0 617.299      .1       0
#XS Ineff= 2 ,-1
   12.69  537.09  139.52  656.56 1023.44   137.8
Permanent Ineff=
       T       T
#Block Obstruct= 8 ,-1
    2.11   62.38  141.16  113.13  141.67  118.96  300.26  308.72     118
  419.74   502.2  131.14  772.86   806.7   137.8  833.13  864.85  128.74
   873.3  903.96  136.36  914.54  963.17  135.46
Bank Sta=582.549,617.299
XS Rating Curve= 0 ,0
Exp/Cntr=0.3,0.1

Type RM Length L Ch R = 5 ,610.5529,,,
BEGIN DESCRIPTION:
E160
END DESCRIPTION:
IW Pilot Flow=0
#Inline Weir SE= 8
       0       0  546.46  110.72  590.88  110.72  593.75  110.69  596.27  110.66
  597.45  110.69  609.23  110.74  615.51  110.74
IW Dist,WD,Coef,Skew,MaxSub,Min_El,Is_Ogee,SpillHt,DesHd
1,3.24,1.7,0,0.98,, 0 ,,,0,0,

Type RM Length L Ch R = 1 ,538.3986,4.268,4.239,4.21
XS GIS Cut Line= 4
529340.4758741344779759.48771593529933.5982441884779827.40540168
530014.5516588064779859.52930789530255.6787853644779678.14392849
#Sta/Elev= 30
       0 112.838  37.388 113.208  44.584 112.201  75.677 111.791 132.671 112.597
 137.186 110.736 171.562  110.81 175.527 112.396  186.54 112.647 222.501 111.626
 302.941 111.746 429.502 112.387 468.339 113.617 473.987  111.92 476.437 113.402
 505.249 114.262 595.159 114.275 596.799  111.47 616.536  111.97 617.003 111.506
 617.477 108.835 625.041 108.565 628.958 108.724  629.46 109.404 629.867 113.521
 630.235     113 727.018 112.885 782.721 114.229 820.314 113.543 979.774 115.933
#Mann= 3 ,-1 , 0
       0      .1       0 616.536    .036       0 630.235      .1       0
Levee=-1,28.19,113.31,0,,,Levee 5,
#XS Ineff= 2 , 0
          597.36  123.62  661.67           125.3
Permanent Ineff=
       T       T
#Block Obstruct= 10 ,-1
   76.65  107.49  116.25  204.41  217.62  117.09  323.35  343.61  131.97
  406.17  426.43  131.79  470.48  493.39  132.95  504.85  597.36  133.56
  675.77  717.18  123.71  835.24  866.08  133.75  875.77  915.42  137.71
  932.16  959.47  137.76
Bank Sta=616.536,630.235
XS Rating Curve= 0 ,0
Exp/Cntr=0.5,0.3

Type RM Length L Ch R = 4 ,536.3362,,,
BEGIN DESCRIPTION:
E161
END DESCRIPTION:
Bridge Culvert--1,0,-1,-1, 0
Deck Dist Width WeirC Skew NumUp NumDn MinLoCord MaxHiCord MaxSubmerge Is_Ogee
0.01,4.04,1.44,0, 18, 18, , , 0.95, 0, ,,,
 596.556  597.11 612.393 615.966 616.414 616.426 616.703 629.614 629.822 631.197
 631.258 631.764 632.957  634.54 637.375 637.378 651.218 651.317
 109.034 109.134 111.906 111.982 111.991 117.049 117.049 117.049 117.049 117.049
 112.061 112.081 112.157 112.269 112.297 112.298 108.336 108.308
 109.034  38.514  38.367  38.333   82.93  84.073 111.623 111.635  38.135  38.142
  38.142  38.144   38.15  38.157   38.17   38.17  38.234 108.308
 597.959 598.513 613.796 617.369 617.817 617.829 618.106 631.017 631.225   632.6
 632.661 633.167  634.36 635.943 638.778 638.781 652.621  652.72
 109.034 109.134 111.906 111.982 111.991 117.049 117.049 117.049 117.049 117.049
 112.061 112.081 112.157 112.269 112.297 112.298 108.336 108.308
 109.034  38.514  38.367  38.333   82.93  84.073 111.623 111.635  38.135  38.142
  38.142  38.144   38.15  38.157   38.17   38.17  38.234 108.308
BR Coef=-1 , 0 , 0 ,, 0 ,,,0.8,-1,,0,
WSPro=,,,, 1 ,,,, 0 ,,,, 0 ,,,,-1 ,-1 ,-1 , 0 , 0 , 0 , 0 , 0
BC Mult= 1 ,0,616,0,617
BC Mult= 3 ,616,631,617,633
BC Mult= 1 ,631,1100,633,1100
BC Design=,, 0 ,, 0 ,,,,,,
BC Use User HTab Curves=0
BC User HTab FreeFlow(D)= 0

Type RM Length L Ch R = 1 ,534.1597,49.546,49.199,48.853
XS GIS Cut Line= 4
529338.7178591254779763.33882777529931.8402291794779831.25651352
530014.4106060734779863.34119268530253.9207703564779681.99504033
#Sta/Elev= 30
       0 124.644    .854 129.001   2.656 132.789  17.164 134.026  18.171 133.262
  19.178 126.726  20.184  113.08  46.141 112.068 134.087 112.487 138.955 110.466
 171.573 112.328 362.324 112.231 372.913 111.877 376.018 110.235 409.713 112.617
 427.655 112.354 431.109  110.64 434.877 112.558 454.736 113.118 618.362 111.884
 619.593 108.818 626.957 108.628 630.633 108.918  631.25  111.93 631.255 112.562
 847.666 115.291 974.526 115.229 983.401 116.176 984.561 118.742 986.003 128.288
#Mann= 3 ,-1 , 0
       0      .1       0 618.362    .036       0 631.255      .1       0
Levee=-1,26.43,113.21,0,,,Levee 5,
#XS Ineff= 2 , 0
          593.83   121.8  666.96          124.55
Permanent Ineff=
       T       T
#Block Obstruct= 11 ,-1
   78.41   96.04  116.62  201.76  220.26  117.93  325.99  360.35  132.77
  409.69  423.79  131.51  470.48  489.87  132.53  509.25  593.83  135.15
  681.06  717.18  123.39   846.7  874.89  133.05  884.58  889.87  133.09
  896.92  921.59  132.77  942.73   967.4  136.87
Bank Sta=618.362,631.25
XS Rating Curve= 0 ,0
Exp/Cntr=0.5,0.3

Type RM Length L Ch R = 1 ,484.9604,50.2,48.985,47.77
XS GIS Cut Line= 5
  529338.7178591 4779763.3388278   529549.483359  4779853.422232
  529891.9278945 4779872.8893995    530011.24978 4779908.0390048
  530256.1909945 4779693.1028995
#Sta/Elev= 30
34.17831133.330544.17062135.211255.16195132.762556.16134126.629157.16056113.0367
 72.1487111.935695.13078112.034898.12852117.1859104.1239115.6292107.1215111.9099
145.0919111.6481147.0905 118.377155.0841121.8044166.0756118.8004179.0655123.1108
193.0545118.5979223.0312 119.099226.0289111.8923 266.796 110.001 561.589 113.637
 580.801 110.365 659.214 111.544 660.263  109.95 667.961 108.709  675.67  111.52
1047.789 115.228 1052.75 117.9171053.458 122.3571054.374 132.6351056.263 135.503
#Mann= 3 ,-1 , 0
34.17831      .1       0 660.263    .036       0  675.67      .1       0
Levee=-1,61.32,112.98,0,,,Levee 5,
#XS Ineff= 2 , 0
          658.68  124.74  684.05          124.09
Permanent Ineff=
       T       T
#Block Obstruct= 9 ,-1
   72.95  207.22  123.71  328.81   356.3  129.92  368.99  519.12  130.25
   566.7  586.78  122.69  639.65  658.68  133.56     683  704.14  123.76
  726.34  772.86  123.15   858.5  890.22  135.38  933.57 1020.26  135.89
Bank Sta=659.214,675.67
XS Rating Curve= 0 ,0
Exp/Cntr=0.5,0.3

Type RM Length L Ch R = 1 ,435.9749,30.271,26.523,25.979
XS GIS Cut Line= 5
  529338.7178591 4779763.3388278  529522.5060944 4779902.5147313
  529716.0253771 4779941.8609755  530033.3876215 4779934.0441714
  530048.1290332 4779932.8157205
#Sta/Elev= 30
-43.0733133.3244-36.1013135.0827-28.1334132.9623-27.1374128.2688-26.1414126.2233
-25.1453116.2209-24.1495 112.983-8.21362111.922550.54966111.669751.54557111.9433
53.53761121.180154.53357122.921659.51349124.611166.48545122.470178.43729125.2399
97.36108 119.512115.2889123.0684131.2247117.9845132.2207113.4812133.2168111.9035
153.1365111.8251160.1084109.4549 300.122 108.655 595.109  111.99 595.289 111.756
 597.339 108.873 602.875 108.602 607.558 109.007   608.6  112.01  716.73 112.326
#Mann= 3 ,-1 , 0
-43.0733      .1       0 595.289    .036       0   608.6      .1       0
#XS Ineff= 2 , 0
          577.97  121.36  632.95          122.04
Permanent Ineff=
       T       T
#Block Obstruct= 6 ,-1
    4.23  112.07  123.48  171.98  177.62   112.2  190.31  229.78   128.6
  253.74  287.58  128.04  307.31  315.07  132.36  338.33  351.72   130.4
Bank Sta=595.109,608.6
XS Rating Curve= 0 ,0
Exp/Cntr=0.5,0.3

Type RM Length L Ch R = 4 ,423.4056,,,
BEGIN DESCRIPTION:
E162
END DESCRIPTION:
Bridge Culvert--1,0,-1,-1, 0
Deck Dist Width WeirC Skew NumUp NumDn MinLoCord MaxHiCord MaxSubmerge Is_Ogee
0.01,26.32,1.44,0, 14, 12, , , 0.95, 0, ,,,
 580.498 580.997 591.594 595.234 595.235 595.325 595.525 608.483 608.787 609.887
 609.893  611.53  628.95 629.111
 109.096 109.233 112.143 112.195 113.296 113.297 113.299 113.412 113.415 113.425
 112.276 112.278 107.896 107.855
 109.096  14.603  14.654  14.671  14.671  14.671 111.517 111.641  14.505  14.511
  14.511   14.52  14.619 107.855
 572.043 575.489 583.139 586.779  586.78  586.87  587.07 600.028 600.332 601.432
 601.438 601.896
 109.096 111.756 112.143 112.195 113.296 113.297 113.299 113.412 113.415 113.425
 112.276 112.278
 109.096  14.603  14.654  14.671  14.671  14.671 111.517 111.641  14.505  14.511
  14.511   14.52
BR Coef=-1 , 0 , 0 ,, 0 ,,,0.8,-1,,0,
WSPro=,,,, 1 ,,,, 0 ,,,, 0 ,,,,-1 ,-1 ,-1 , 0 , 0 , 0 , 0 , 0
BC Mult= 1 ,-200,595,-200,575
BC Mult= 3 ,595,610,575,602
BC Mult= 1 ,610,800,602,800
BC Design=,, 0 ,, 0 ,,,,,,
BC Use User HTab Curves=0
BC User HTab FreeFlow(D)= 0
